HEC-RAS study NFKCHERRYRV.prj: NFKCHERRYRV

--- NFKCHERRYRV.g01 (geometry) --- (continued)

Type RM Length L Ch R = 1 ,54490   ,430.5,435.8,435.7
XS GIS Cut Line= 2
     2134281.078      445098.487     2133153.534      445444.763
#Sta/Elev= 30
       0 3334.03    45.9 3310.74   101.6 3277.79   127.8 3261.69     154 3241.37
   170.4 3237.85     190 3227.82   278.5 3167.13   350.6 3122.95   425.9 3085.58
     593 3011.46   632.4 2999.15   658.6 2996.84     688 2980.53     711  2978.6
   733.9 2978.63   740.5 2981.72     747 2989.45  755.77 2994.51  786.67 2996.69
   799.4 2994.83  817.56 2981.83   845.3  2981.9   887.9 3010.17   937.1 3053.72
   979.6 3082.38  1045.2 3113.96  1100.9 3153.76  1156.6 3171.84  1179.5 3184.19
#Mann= 6 ,-1 , 0
       0     .12       0     688     .04       0   740.5     .12       0
  755.77     .08       0  786.67    .016       0  817.56     .12       0
#XS Ineff= 2 , 0
                          787.56         2997.24
Permanent Ineff=
       F       F
Bank Sta=688,740.5
XS Rating Curve= 0 ,0
Exp/Cntr=0.3,0.1

Type RM Length L Ch R = 1 ,54055   ,557.2,575.3,582.8
XS GIS Cut Line= 2
2134117.19112302 444757.167531382133087.17722894444976.678689136
#Sta/Elev= 30
       0 3264.11    34.7 3252.02    57.9 3237.06   111.9 3209.85   199.1 3159.53
   269.5 3134.22   326.6 3107.36     350 3093.88   473.1 3037.55   487.6 3027.01
   521.1 3010.38   567.1 2980.72   578.1 2978.18   611.7 2979.49     6212975.043
   628.4 2972.66   665.3 2972.38   680.5 2975.07   698.9 2989.37   705.4  2990.5
   735.8 2990.34   762.6 2975.31   786.1 2976.97   816.3 3005.16   846.6  3026.7
   876.7 3053.41     919 3081.14   957.2 3102.23   990.7 3127.14  1053.1 3163.05
#Mann= 3 , 0 , 0
       0     .12       0     621     .04       0   680.5     .12       0
#XS Ineff= 2 , 0
                          726.52         2991.95
Permanent Ineff=
       F       F
Bank Sta=621,680.5
XS Rating Curve= 0 ,0
Exp/Cntr(USF)=0,0
Exp/Cntr=0.3,0.1

Type RM Length L Ch R = 1 ,53479   ,780,775.1,775.8
XS GIS Cut Line= 4
     2134206.671      444288.602     2133605.696      444377.317
     2133448.298       444317.22     2132964.656      444371.594
#Sta/Elev= 30
       0 3373.08    52.3 3337.22   137.2 3291.94     160 3275.53   179.6 3268.08
   238.4 3238.36   313.5 3189.11   372.3 3154.19   431.1 3126.49   512.8 3080.53
   558.5 3042.61   597.7 3015.69     614 3000.63   633.4  2987.7   652.8 2971.44
     669 2965.53     695 2964.04   711.2 2962.33   730.6 2964.03   743.6 2967.95
   772.7 2969.85   860.9 2967.86   880.5 2971.94  902.74 2982.04  932.46 2985.18
   952.4 2985.17   994.8 3017.64  1043.8 3040.29  1138.5 3076.88  1262.7 3141.69
#Mann= 5 ,-1 , 0
       0     .12       0     695     .04       0   730.6     .12       0
  902.74    .016       0  932.46     .12       0
#XS Ineff= 2 , 0
                          781.91         2970.35
Permanent Ineff=
       F       F
Bank Sta=695,730.6
XS Rating Curve= 0 ,0
Exp/Cntr=0.3,0.1

Type RM Length L Ch R = 1 ,52704   ,360.6,348.6,335.6
XS GIS Cut Line= 2
      2134043.55       443533.09     2132818.705      443736.277
#Sta/Elev= 30
       0 3301.72    75.4 3274.79   137.6 3245.36   157.2 3233.64   242.4 3195.19
   294.8  3156.3   340.7 3130.69   370.2 3118.01   393.1 3103.91   484.8  3057.3
   530.7 3025.09   599.5 3007.42     629 2996.71   661.7 2994.26   710.9 2973.74
   743.6 2954.73   789.5 2956.68   802.6  2951.8   815.7 2949.74   861.6 2950.96
   887.8 2967.54  910.73 2967.78   930.4 2965.94  940.67 2970.39   966.4  2989.6
   989.3 3002.45  1018.8 3014.63  1120.4 3070.29  1182.6 3113.63  1241.6 3151.07
#Mann= 5 ,-1 , 0
       0     .12       0   802.6     .04       0   861.6     .12       0
  910.73    .016       0  940.67     .12       0
#XS Ineff= 2 , 0
          783.97 2968.85
Permanent Ineff=
       F       F
Bank Sta=802.6,861.6
XS Rating Curve= 0 ,0
Exp/Cntr=0.3,0.1

Type RM Length L Ch R = 1 ,52356   ,194.2,173.5,169.8
XS GIS Cut Line= 3
2133703.53174925443282.6851582462133286.16695036443247.639259103
 2132719.0605824443566.238342226
#Sta/Elev= 30
       0 3116.41    48.8 3094.12   129.3 3045.42     149 3041.87   185.2 3028.43
   234.6 3018.25   287.3 3001.59   392.1 2979.06   412.4 2971.45   445.1 2948.72
   565.6 2946.31   598.8 2945.56   642.62948.056   679.2 2959.76   702.9 2972.33
   727.6  2972.4   746.4 2971.72     768 2992.04   776.5 2999.15   794.5 3007.19
   814.1 3025.92   866.8 3060.59   906.9 3094.17     912 3102.14   915.7  3111.1
   930.8 3158.74   934.6 3167.54   999.3 3183.37  1024.9 3196.45  1069.3 3227.33
#Mann= 5 ,-1 , 0
       0     .12       0   565.6     .04       0   642.6     .12       0
   727.6    .016       0     768     .12       0
Bank Sta=565.6,642.6
XS Rating Curve= 0 ,0
Exp/Cntr(USF)=0,0
Exp/Cntr=0.3,0.1

Type RM Length L Ch R = 1 ,52182   ,323.9,328.1,314.3
XS GIS Cut Line= 3
2133442.28050109442712.3927994552133095.00750048443139.315570841
2132684.01468325443496.146543939
#Sta/Elev= 30
       0 3081.21    97.3  3047.7   228.4 3007.86   419.2 2973.82   431.4 2966.23
   445.2 2962.09     461 2951.85   472.6  2947.1   495.9 2945.08   547.2 2945.46
   571.1 2942.04   627.6 2942.86   649.3 2945.88   701.4 2952.62   749.9  2976.1
   777.5 2976.73   798.4 2975.14   810.1 2980.88   831.8 2994.31     855 3000.66
   882.1 3020.89     897 3038.93   920.1 3052.63   975.2  3092.2    1003 3118.29
    1024 3135.13  1040.3 3164.14  1050.2 3173.65  1083.8 3192.37  1094.6 3200.64
#Mann= 5 ,-1 , 0
       0     .12       0   547.2     .04       0   649.3     .12       0
   777.5    .016       0   810.1     .12       0
Bank Sta=547.2,649.3
XS Rating Curve= 0 ,0
Exp/Cntr(USF)=0,0
Exp/Cntr=0.3,0.1

Type RM Length L Ch R = 1 ,51854   ,1041.9,1029.8,995.4
XS GIS Cut Line= 4
     2133013.307       442331.14     2132941.762      442834.815
     2132795.811      443046.587     2132606.933      443441.513
#Sta/Elev= 30
       0 3183.83    45.7 3161.34   104.4 3141.77   290.2 3072.54   463.1 2993.04
   479.4  2988.2   508.7 2986.23   564.1 2971.54   573.8 2965.96   609.6 2937.02
   629.2 2935.45   671.5 2937.03   697.6 2939.02   720.4 2936.31   746.4 2939.47
   756.2 2944.25   788.8    2945   811.7 2950.32  869.34 2976.33  914.78 2974.15
   922.7 2973.85  934.82 2982.03   958.7 3004.62  1043.6 3052.78  1076.3 3074.62
  1089.4  3084.5  1115.5 3114.86  1154.7 3141.19  1174.3 3164.65  1203.7 3177.37
#Mann= 6 ,-1 , 0
       0     .12       0   609.6     .04       0   671.5     .12       0
  869.34    .016       0  914.78     .06       0  934.82     .12       0
Bank Sta=609.6,671.5
XS Rating Curve= 0 ,0
Exp/Cntr=0.3,0.1

Type RM Length L Ch R = 1 ,50824   ,579.6,588.3,589.8
XS GIS Cut Line= 4
     2131860.007       442362.62     2131940.137      442920.668
     2132003.097      443255.497     2132091.812      443570.294
#Sta/Elev= 30
       0 3256.49    22.9 3242.54    68.8 3220.84   127.8 3206.34   147.5  3197.7
   170.4 3181.83   193.4 3150.22     213 3137.58   232.7 3120.93   288.4 3085.05
   344.2 3053.67   452.3 3005.65   514.6 2982.56   593.3 2958.68   639.1 2939.13
   655.5 2929.79   675.2 2927.24   691.5 2919.45   740.7 2917.64   753.8 2919.13
   770.2 2922.96   793.1 2924.18  816.88 2934.42  850.82 2936.05   865.2 2934.75
   878.3 2929.58   907.7 2931.96  1005.9 2991.58  1120.3 3053.32  1231.5 3118.73
#Mann= 5 ,-1 , 0
       0     .12       0   691.5     .04       0   753.8     .12       0
  816.88    .016       0  850.82     .12       0
Bank Sta=691.5,753.8
XS Rating Curve= 0 ,0
Exp/Cntr=0.3,0.1

Type RM Length L Ch R = 1 ,50236   ,903,913.1,907.5
XS GIS Cut Line= 3
     2131590.999      442499.986     2131402.122      443000.798
     2131425.016      443659.009
#Sta/Elev= 30
       0 3192.64    39.2 3184.16    94.6 3177.54     111 3161.17   133.8    3157
   150.1 3145.36   195.8 3120.81   218.7 3103.67   267.6 3073.58   323.1 3050.83
   398.2 3009.94   443.9 2995.15     483 2978.37     568 2919.16   672.9 2919.45
   718.7 2915.04   725.3 2912.33   735.1 2909.25   754.8 2908.86     781 2911.09
   800.7 2923.63  822.19 2926.24   843.2 2927.92  851.74 2933.41   859.6 2940.41
   882.6 2952.81   961.2  2977.5  1026.7 2988.89  1069.3 3003.19  1193.8 3075.34
#Mann= 5 ,-1 , 0
       0     .12       0   725.3     .04       0     781     .12       0
  822.19    .016       0  851.74     .12       0
Bank Sta=725.3,781
XS Rating Curve= 0 ,0
Exp/Cntr=0.3,0.1

Type RM Length L Ch R = 1 ,49323   ,1013.6,1009.9,985.1
XS GIS Cut Line= 4
     2130569.342      442236.702      2130549.31      442883.465
     2130537.862      443238.326     2130586.513      443636.115
#Sta/Elev= 30
       0 3188.63    55.6 3164.64   163.4 3103.67   277.8 3058.47     317 3045.37
   349.7 3037.71     415 3015.02   545.8 2961.79     585 2948.73   614.4 2936.73
   656.8 2908.69   673.1 2904.76     748 2905.42  759.42 2897.38   783.9 2895.77
   809.9 2897.43     937 2903.24   966.3 2918.44   982.6 2911.73  992.28 2910.84
  1015.2 2909.34 1021.97 2912.19  1034.7 2923.36    1051 2931.13  1083.6 2954.73
    1139 2977.27  1233.4 3024.62  1327.9 3097.02  1350.7 3129.66  1402.9 3145.89
#Mann= 5 ,-1 , 0
       0     .12       0  759.42     .04       0   809.9     .12       0
  992.28    .016       0 1021.97     .12       0
Bank Sta=759.42,809.9
XS Rating Curve= 0 ,0
Exp/Cntr=0.3,0.1

Type RM Length L Ch R = 1 ,48313   ,852.1,843.8,831.3
XS GIS Cut Line= 3
     2129473.278      443106.684     2129825.278      443704.798
     2130074.253      443953.773
#Sta/Elev= 30
       0 3026.44      36 3011.88    81.8 2985.83     144 2959.68     180 2939.67
   199.7 2924.65   261.9 2886.13   288.1  2884.3   324.1 2886.57   337.2 2884.92
   441.9 2887.17     478 2883.92   487.8 2880.85   510.7 2879.51   540.2 2880.88
   569.6 2885.81     622 2883.37     658 2884.46   697.3 2896.14  710.64 2894.76
   742.9 2894.38  752.41 2898.36   762.5 2907.45   772.2 2921.53     782 2931.72
   804.8 2948.96   889.6 2990.85   971.1 3039.47  1023.3  3067.7  1046.1 3083.22
#Mann= 5 ,-1 , 0
       0     .12       0   487.8     .04       0   540.2     .12       0
  710.64    .016       0  752.41     .12       0
#XS Ineff= 2 , 0
          440.48 2909.42  599.91         2884.91
Permanent Ineff=
       F       F
Bank Sta=487.8,540.2
XS Rating Curve= 0 ,0
Exp/Cntr=0.3,0.1

Type RM Length L Ch R = 1 ,47469   ,482.1,483.7,479.3
XS GIS Cut Line= 2
     2128809.344      443827.854     2129713.668      444531.854
#Sta/Elev= 30
       0 3060.95    22.9 3044.86    32.7 3042.39    65.5 3021.31   137.5  2990.2
   163.7  2971.1   186.6 2963.57   206.3 2952.67   245.6 2924.34     262 2915.74
   288.2  2887.1   304.5 2877.01   376.6  2871.2   435.5 2873.66   586.1 2870.82
   605.8 2873.06   638.5 2866.98   651.6 2865.47   690.9 2867.47  707.19 2878.67
  740.93 2882.46   772.8 2882.93  778.36 2886.17   802.2 2911.73   841.5 2945.38
   887.4 2961.12     907  2972.7   988.9 3009.79  1083.8 3065.55    1146 3097.33
#Mann= 6 ,-1 , 0
       0     .12       0   638.5     .04       0   690.9     .12       0
  707.19     .08       0  740.93    .016       0  778.36     .12       0
#XS Ineff= 2 , 0
          603.73 2882.71
Permanent Ineff=
       F       F
Bank Sta=638.5,690.9
XS Rating Curve= 0 ,0
Exp/Cntr=0.3,0.1

Type RM Length L Ch R = 1 ,46985   ,446.7,455.7,444.2
XS GIS Cut Line= 2
2128481.66428449444170.3973212252129423.02944179444900.694057605
#Sta/Elev= 30
       0 3121.77    30.6 3102.26    72.1 3071.76   109.5 3054.67   182.3 3009.77
     259    2967   296.9 2955.93   335.1 2936.98   411.5 2905.46   433.4 2899.63
   474.3 2894.63   516.4 2862.78   544.8  2861.1   574.6 2863.61   599.5  2861.2
     667 2864.01   698.52858.537   708.5 2857.44   754.12859.026   762.2 2860.65
   779.4 2872.45   790.3 2874.49   820.7 2874.34   840.3 2864.84   854.3 2864.44
   898.4  2896.1   921.2 2907.96   948.3 2918.62   984.4  2925.8  1191.4 3031.69
#Mann= 3 , 0 , 0
       0     .12       0   698.5     .04       0   754.1     .12       0
Bank Sta=698.5,754.1
XS Rating Curve= 0 ,0
Exp/Cntr(USF)=0,0
Exp/Cntr=0.3,0.1

Type RM Length L Ch R = 1 ,46530   ,912.3,925.4,924.7
XS GIS Cut Line= 2
     2128231.263      444531.854     2129061.181      445170.032
#Sta/Elev= 30
       0 3097.67    29.4 3076.11    55.6 3063.63    65.4 3056.09   124.3 3024.06
   196.3 2988.39   212.6 2976.77   258.5 2950.24   278.1 2943.58     301 2940.02
   327.2 2930.62   353.3 2925.64   382.8 2914.09   474.4  2857.2   484.2 2854.46
   520.2 2854.16   533.3    2851   621.6 2856.01   654.3  2853.5   713.2 2853.72
   742.7 2856.74   755.7 2864.47   769.1 2866.28     795 2867.56   808.1 2865.32
  817.55 2869.99   906.2 2924.66   981.5 2948.04  1017.5 2964.34  1046.9 2974.14
#Mann= 5 ,-1 , 0
       0     .12       0   654.3     .04       0   713.2     .12       0
   769.1    .016       0  817.55     .12       0
Bank Sta=654.3,713.2
XS Rating Curve= 0 ,0
Exp/Cntr=0.3,0.1

Type RM Length L Ch R = 1 ,45604   ,826.6,832.4,829.9
XS GIS Cut Line= 3
     2127676.077      444995.463     2128091.036      445479.105
     2128319.979      445802.486
#Sta/Elev= 30
       0  3036.1    32.7 3021.58   114.4 2994.46   235.3    2940   271.2    2932
   310.5 2905.95   336.6 2878.44   352.9 2866.32   382.4  2838.5   388.9 2834.41
   398.7 2833.79   447.7 2834.34   467.3 2839.91   486.9 2840.92     500 2840.31
   506.5 2836.42   558.8 2835.76   578.4  2840.8   719.1 2843.42   735.5 2850.59
  745.33 2851.61   771.5 2850.92  796.45 2838.92   840.3 2845.81   869.8 2861.24
   954.9 2889.58   981.1 2903.05  1007.3 2905.18 1028.18 2919.77  1033.5 2922.59
#Mann= 6 ,-1 , 0
       0     .12       0   506.5     .04       0   558.8     .12       0
  745.33    .016       0  796.45     .12       0 1028.18    .016       0
#XS Ineff= 2 , 0
             480 2842.38  744.43         2879.83
Permanent Ineff=
       F       F
Bank Sta=506.5,558.8
XS Rating Curve= 0 ,0
Exp/Cntr=0.3,0.1

Type RM Length L Ch R = 1 ,44772   ,716.5,707.8,670
XS GIS Cut Line= 3
     2127109.443      445467.657     2127561.605      446091.527
     2127707.557      446309.022
#Sta/Elev= 30
       0 2944.84    68.8 2915.56   239.4 2858.75   295.1 2835.17     318 2832.08
   383.6 2831.91   403.3 2828.74   465.6 2828.72   495.1  2823.7   557.4 2826.46
   619.7 2822.46   629.5 2821.72   668.9 2823.25   671.8  2824.5   691.8 2835.82
  700.01 2836.52  736.49 2833.33   750.8 2829.03   770.5 2828.66     800 2834.47
   813.1 2840.34   842.5 2863.73     872  2901.7   891.6 2913.09   914.6 2930.32
   927.6 2942.06   940.8 2957.63   950.6 2961.84   999.7 3001.14  1032.4 3019.61
#Mann= 6 ,-1 , 0
       0     .12       0   619.7     .04       0   668.9     .12       0
   671.8     .08       0  700.01    .016       0  736.49     .12       0
Bank Sta=619.7,668.9
XS Rating Curve= 0 ,0
Exp/Cntr=0.3,0.1

Type RM Length L Ch R = 1 ,44064   ,562.9,559.7,542.5
XS GIS Cut Line= 4
     2126436.924      446317.608     2126786.062      446383.429
     2127100.858      446466.421     2127346.972      446592.339
#Sta/Elev= 30
       0 2932.14      88 2901.72     176 2863.72     189    2862   241.2 2844.86
   309.6 2819.73   322.7 2818.99   342.2 2826.51   368.3 2818.14   381.3 2816.41
     492 2817.13   527.8 2814.47   592.9 2814.01  608.45 2813.25  608.71 2813.24
   625.5 2812.31     658 2814.82   690.6 2813.28   713.4 2824.13   735.2 2825.62
  768.38 2825.15   791.4 2821.64  801.56 2827.93   820.7 2841.18   833.7 2858.82
     850 2874.78   859.7 2890.58   866.2 2898.27   918.3 2946.62   957.3 2965.27
#Mann= 8 ,-1 , 0
       0     .12       0   527.8     .04       0   592.9     .12       0
  608.45     .08       0  608.71     .12       0   735.2     .08       0
  768.38    .016       0  801.56     .12       0
#XS Ineff= 2 , 0
          497.55 2816.71
Permanent Ineff=
       F       F
Bank Sta=527.8,592.9
XS Rating Curve= 0 ,0
Exp/Cntr=0.3,0.1

Type RM Length L Ch R = 1 ,43504   ,412.4,405.6,392.1
XS GIS Cut Line= 4
     2126594.322      446984.404     2126952.045        446947.2
     2127129.476      446967.233     2127292.598      446927.168
#Sta/Elev= 30
       0 2888.53    19.6 2883.16    55.6 2876.13      85 2872.18   143.9 2859.48
   163.5 2853.17   176.6 2845.71   199.4  2835.9   238.7 2825.44   261.6 2813.88
   281.2  2809.4   343.3 2808.61   379.1 2803.73   431.1 2804.17   447.3 2802.18
   463.5 2801.29   476.5 2802.53   486.3 2807.01   499.2 2808.94   544.7 2806.16
   589.9 2806.86   609.3 2815.24  619.41 2815.06     648 2811.28     661 2812.68
   667.4 2815.48  680.23 2825.32   686.8 2831.34   699.7 2836.76   706.2 2841.72
#Mann= 5 ,-1 , 0
       0     .12       0   447.3     .04       0   476.5     .12       0
  619.41    .016       0  680.23     .12       0
#XS Ineff= 2 , 0
                          522.36         2807.56
Permanent Ineff=
       F       F
Bank Sta=447.3,476.5
XS Rating Curve= 0 ,0
Exp/Cntr=0.3,0.1

Type RM Length L Ch R = 1 ,43099   ,752.3,761.4,749.8
XS GIS Cut Line= 2
     2126860.468      447553.899     2127449.996      447075.981
#Sta/Elev= 30
       0 2957.98    78.5 2922.79    94.9  2917.8   186.5 2880.89   215.9 2868.21
   255.2  2848.4   271.5 2845.62   310.8  2827.7   320.6 2826.29   340.2 2818.16
   382.7  2807.4   408.9 2803.85   448.2 2800.01   484.1  2802.9   503.8 2797.13
   526.7 2795.25     543 2794.17   572.5 2794.32     579 2796.52   585.5 2800.32
   601.9 2802.95   611.7  2809.1  630.52 2809.05   647.7 2807.75   660.8 2803.17
  675.95 2802.67   693.5  2803.8   703.3 2807.17   726.2 2829.27   758.9 2855.32
#Mann= 5 ,-1 , 0
       0     .12       0   526.7     .04       0     579     .12       0
  630.52    .016       0  675.95     .12       0
#XS Ineff= 2 , 0
          482.53 2803.07
Permanent Ineff=
       F       F
Bank Sta=526.7,579
XS Rating Curve= 0 ,0
Exp/Cntr=0.3,0.1

Type RM Length L Ch R = 1 ,42337   ,701.3,705.4,694
XS GIS Cut Line= 2
     2127352.695      448129.118     2128045.247      447545.314
#Sta/Elev= 30
       0  3015.7    58.9 2987.93   117.7 2958.08   143.9 2941.12   153.7 2936.42
   258.3 2904.76   330.3 2874.76   343.4    2871   402.2 2837.39   428.4 2810.58
   454.5 2791.27   464.3  2789.7   480.7 2789.97   493.8 2786.21   523.2 2786.21
   565.7 2784.81   585.3 2786.12   608.2 2797.22  622.43 2798.42   644.2 2797.77
  661.06 2790.29   673.6 2785.33   696.5 2785.45   758.6 2793.42   794.6 2816.34
   804.4 2819.17   837.1 2837.32   856.7 2846.36     896 2868.65   905.8 2871.96
#Mann= 5 ,-1 , 0
       0     .12       0   523.2     .04       0   585.3     .12       0
  622.43    .016       0  661.06     .12       0
#XS Ineff= 2 , 0
           483.7 2815.19  623.52          2812.3
Permanent Ineff=
       F       F
Bank Sta=523.2,585.3
XS Rating Curve= 0 ,0
Exp/Cntr=0.3,0.1

Type RM Length L Ch R = 1 ,41632   ,912.8,912.7,896.8
XS GIS Cut Line= 2
     2127764.792      448707.199     2128471.653      448028.955
#Sta/Elev= 30
       0 3078.06      36  3055.9     118 3000.04   137.6 2984.15     154 2965.21
   193.3 2938.11     249 2913.18   262.1 2910.39   301.4 2891.05   317.8 2886.92
   350.6 2871.32   429.2 2822.93   458.7 2792.96   478.4 2777.12   527.5 2775.11
   553.7 2776.96   573.4 2775.96   583.2 2781.73   589.7 2782.75   671.6 2779.02
   684.8 2780.96  703.49 2788.05  746.16 2785.91   773.2 2784.81   789.6 2787.51
     806 2785.92   828.9 2791.23   887.9 2798.44   946.9  2812.6   979.6 2826.74
#Mann= 5 ,-1 , 0
       0     .12       0   478.4     .04       0   553.7     .12       0
  703.49    .016       0  746.16     .12       0
#XS Ineff= 2 , 0
                          658.55         2780.45
Permanent Ineff=
       F       F
Bank Sta=478.4,553.7
XS Rating Curve= 0 ,0
Exp/Cntr=0.3,0.1

Type RM Length L Ch R = 1 ,40719   ,738.4,780.1,797.4
XS GIS Cut Line= 4
      2128563.23      449205.149     2128700.596      449064.922
       2128835.1      448887.491      2129204.27       448469.67
#Sta/Elev= 30
       0 2913.66    13.1 2908.76    26.2 2896.86    39.3 2888.31    58.9 2889.04
      72 2884.46    91.6 2872.78   114.5 2855.19   137.4 2834.25   179.9 2807.17
     193 2794.88   258.5 2767.52   330.5 2764.67   346.9 2767.57     360 2770.75
   415.2 2771.79  442.38 2771.91  481.79 2772.03  521.21  2770.9   540.3  2770.4
  549.35 2773.64  560.62 2776.16   582.9 2776.51  600.04 2770.04   697.7 2772.66
   845.3 2770.19     865 2774.16   927.3 2800.55  954.76 2808.03   976.5 2807.41
#Mann= 11 ,-1 , 0
       0     .12       0   258.5     .04       0   346.9     .12       0
   415.2     .06       0  442.38     .12       0  481.79    .016       0
  521.21     .06       0  549.35     .08       0  560.62    .016       0
  600.04     .12       0  954.76    .016       0
#XS Ineff= 2 , 0
                          473.15         2783.63
Permanent Ineff=
       F       F
Bank Sta=258.5,346.9
XS Rating Curve= 0 ,0
Exp/Cntr=0.3,0.1

Type RM Length L Ch R = 1 ,39939   ,921.4,953.2,960.7
XS GIS Cut Line= 3
     2128577.539      449291.003      2129347.36      449517.084
     2130100.009      449963.522
#Sta/Elev= 30
       0 2891.65    29.5 2873.68    62.2 2833.46   111.3 2779.44   124.4 2771.54
   150.6 2762.87   163.7  2759.4   232.5 2759.68   248.9 2756.26   268.5 2759.29
     393 2760.89   415.9 2756.08   533.8 2760.94   717.2 2758.07     763 2759.39
   769.6 2765.59  789.41 2767.57   808.9 2768.33  822.25 2763.62   844.9 2758.43
   864.6 2765.82  1025.2 2773.51  1071.1 2770.43  1126.8 2775.15  1192.4 2773.71
  1284.1 2786.13  1395.6 2792.61  1503.7 2803.58  1644.6 2821.54  1677.4 2829.41
#Mann= 5 ,-1 , 0
       0     .12       0   717.2     .04       0     763     .08       0
  789.41    .016       0  822.25     .12       0
#XS Ineff= 2 , 0
           452.6 2769.05  801.81         2768.34
Permanent Ineff=
       F       F
Bank Sta=717.2,763
XS Rating Curve= 0 ,0
Exp/Cntr=0.3,0.1

Type RM Length L Ch R = 1 ,38986   ,358.3,357.4,356
XS GIS Cut Line= 2
     2128357.182      449528.531     2128889.474      450450.026
#Sta/Elev= 30
       0 2843.43   140.8  2787.2   229.2 2760.29   268.5 2753.29   399.5 2749.24
   415.8  2750.9   484.6 2750.58     537 2745.72   569.8 2746.35   605.8 2742.96
   635.2 2745.27   661.4 2743.99   674.5 2741.26   694.2 2740.05   723.6 2741.36
   749.8 2748.35   762.9 2753.78  808.47 2756.17   821.9 2756.79     835 2768.62
  842.58 2771.72   867.7 2779.74   884.1 2780.61   897.2 2787.27   910.3 2798.42
   923.4 2802.76   985.6 2797.26   998.7 2798.65  1034.7 2819.38  1064.2 2828.36
#Mann= 5 ,-1 , 0
       0     .12       0   674.5     .04       0   723.6     .12       0
  808.47    .016       0  842.58     .12       0
#XS Ineff= 2 , 0
           551.5 2747.09
Permanent Ineff=
       F       F
Bank Sta=674.5,723.6
XS Rating Curve= 0 ,0
Exp/Cntr=0.3,0.1

Type RM Length L Ch R = 1 ,38628   ,614.1,626,640.4
XS GIS Cut Line= 2
     2128072.994      449818.544     2128607.175      450619.816
#Sta/Elev= 30
       0 2791.24      36 2782.89    65.5 2778.39   140.8 2773.91   160.5 2771.19
   209.6  2748.4   229.3 2743.85   360.3 2743.62   383.2 2742.78   402.9 2739.67
   429.1 2744.26   491.3 2742.34   556.8 2743.99   596.2 2740.56   602.7 2737.67
   612.5 2735.97   638.7 2737.54   658.4 2738.83   674.8 2737.56   687.9 2742.85
     701 2744.32   714.1 2749.79   743.6 2752.56   759.9  2750.5   766.5 2751.71
   786.1 2762.64   799.2 2772.25   861.5 2783.26   913.9 2809.04     963 2830.55
#Mann= 3 , 0 , 0
       0     .12       0   602.7     .04       0   638.7     .12       0
#XS Ineff= 2 , 0
           557.8 2745.85
Permanent Ineff=
       F       F
Bank Sta=602.7,638.7
XS Rating Curve= 0 ,0
Exp/Cntr=0.3,0.1

Type RM Length L Ch R = 1 ,38002   ,717.4,710.9,681.2
XS GIS Cut Line= 3
     2127847.784       449831.88     2127844.922      450570.221
      2127842.06      450816.334
#Sta/Elev= 30
       0  2820.9   137.2 2771.23   192.8 2755.18   209.1 2747.78   241.8 2737.76
     294 2736.27   320.2 2733.88   356.1 2737.86   362.6    2737   375.7 2731.43
     392 2730.18   450.8 2732.49   499.8 2730.84   532.5 2734.26   614.2 2734.17
   637.1 2730.28   646.9 2729.05   699.1 2730.62  721.63 2746.38   728.6 2748.84
  751.17 2749.34   764.2  2746.6   767.5 2747.41   777.2 2755.13   790.2  2768.6
   796.6 2776.99   803.1 2781.69     829 2789.89   903.5 2824.76   984.5  2853.1
#Mann= 5 ,-1 , 0
       0     .12       0   637.1     .04       0   699.1     .12       0
  721.63    .016       0  751.17     .12       0
#XS Ineff= 2 , 0
          534.68  2742.2
Permanent Ineff=
       F       F
Bank Sta=637.1,699.1
XS Rating Curve= 0 ,0
Exp/Cntr=0.3,0.1

Type RM Length L Ch R = 1 ,37292   ,414.3,416.8,407.3
XS GIS Cut Line= 3
     2127143.785      449886.254     2127284.012      450355.587
     2127358.419      450681.831
#Sta/Elev= 30
       0  2878.5    29.4 2857.48    55.5 2851.83    71.8 2845.56   117.6    2818
   130.6 2814.97   169.8 2812.61   195.9 2808.53   212.3 2803.21   228.6 2795.35
   248.2 2781.66   267.8 2772.48   329.8 2724.56   339.6 2720.65   404.9 2719.45
   414.7 2720.89   444.1 2725.31     467 2722.14   493.1  2724.7   578.4 2724.06
   637.5 2726.91   663.7 2733.07   680.1 2741.17   699.8 2746.77   716.2 2756.82
  723.13 2758.73   765.4 2755.62  783.72 2770.88   794.9 2778.72   824.4 2789.91
#Mann= 5 ,-1 , 0
       0     .12       0   339.6     .04       0   414.7     .12       0
  723.13    .016       0  783.72     .12       0
#XS Ineff= 2 , 0
                          439.31         2731.22
Permanent Ineff=
       F       F
Bank Sta=339.6,414.7
XS Rating Curve= 0 ,0
Exp/Cntr=0.3,0.1

Type RM Length L Ch R = 1 ,36875   ,531.7,522.4,516.7
XS GIS Cut Line= 2
 2126738.2391277450059.2062648622127088.61270642450937.250895885
#Sta/Elev= 30
       0 2897.23    20.1 2888.57    34.2 2878.76    44.8 2875.65    76.6 2855.84
      87 2852.59    94.6 2846.48   127.4 2832.51   161.4 2812.26   175.4  2808.6
   200.3  2796.8   273.8 2747.72   313.3 2717.12   352.1 2717.41   359.7 2714.08
   408.7 2712.58   429.9 2713.27   440.4 2718.45   453.1  2720.1     550 2720.47
   578.2  2717.5   613.6 2722.71   624.2 2727.72   642.5  2729.2   708.9  2743.7
   737.2 2758.43     776 2755.08   800.8  2766.3   878.5  2791.8   945.4 2810.74
#Mann= 3 , 0 , 0
       0     .12       0   359.7     .04       0   429.9     .12       0
#XS Ineff= 2 , 0
                          548.89         2742.74
Permanent Ineff=
       F       F
Bank Sta=359.7,429.9
XS Rating Curve= 0 ,0
Exp/Cntr(USF)=0,0
Exp/Cntr=0.3,0.1

Type RM Length L Ch R = 1 ,36352   ,592.6,579.2,566.5
XS GIS Cut Line= 3
     2126233.737       450392.79     2126491.298      450721.896
     2126826.127      451079.619
#Sta/Elev= 30
       0  2831.9    65.3 2814.33    91.4  2803.6   104.5 2803.03   124.1 2793.38
   140.4 2789.32     160  2776.2   202.4  2734.1   225.3 2715.11   257.9 2708.32
   303.6 2706.69     320 2707.65   378.7 2711.85   427.7 2708.88   447.3 2710.35
     480 2708.88     493 2711.56   515.9 2711.72     529 2715.46   656.4  2712.3
   672.7 2717.54   751.1 2718.67   760.9 2720.37     774 2726.42   800.1 2746.59
  818.89 2747.88   849.1 2745.32  862.11 2750.14   901.4 2783.05   907.9 2786.54
#Mann= 5 ,-1 , 0
       0     .12       0   257.9     .04       0     320     .12       0
  818.89    .016       0  862.11     .12       0
#XS Ineff= 2 , 0
                          529.35         2716.06
Permanent Ineff=
       F       F
Bank Sta=257.9,320
XS Rating Curve= 0 ,0
Exp/Cntr=0.3,0.1

Type RM Length L Ch R = 1 ,35773   ,525.1,510.5,497.2
XS GIS Cut Line= 3
     2125921.802      451005.212     2126273.802       451145.44
     2126631.525      451311.423
#Sta/Elev= 30
       0 2802.76    39.2 2790.58    62.1 2781.85    71.9  2776.1    88.2 2772.65
   120.9 2756.07     147 2738.18   166.6 2722.36   189.4 2707.98   212.3 2701.19
   225.4 2700.52   287.4 2701.38   303.8 2709.43   310.3  2711.2     356 2711.45
   385.4 2709.89   414.8 2712.12   444.1 2709.59   463.6 2714.36   486.4  2714.8
   587.5 2711.06   620.1  2713.3   688.5 2712.35   704.8 2716.28   724.4 2731.26
   730.9 2734.44   737.4 2735.57  757.94 2735.67   766.7 2734.96   773.3  2737.2
#Mann= 4 ,-1 , 0
       0     .12       0   212.3     .04       0   287.4     .12       0
  757.94    .016       0
Bank Sta=212.3,287.4
XS Rating Curve= 0 ,0
Exp/Cntr=0.3,0.1

Type RM Length L Ch R = 1 ,35263   ,762.9,777.5,779.2
XS GIS Cut Line= 3
     2125964.729      451586.155     2126248.046      451574.708
     2126502.745      451660.561
#Sta/Elev= 30
       0 2750.42     9.8 2746.25    26.1  2743.9    39.1 2738.19    78.2 2725.87
   104.3 2719.77   117.3 2714.24   127.1 2707.14   133.6 2703.57   149.9 2697.33
   156.4  2696.5   195.6  2696.1   215.1 2695.62   228.1 2697.43   247.7 2705.88
   273.8 2703.45   290.1 2705.64   316.3 2704.54   368.8 2704.56   408.1 2707.28
   414.7 2708.94   421.2 2711.89   434.3 2719.82   447.4 2729.32  455.38 2731.63
   483.5 2731.47   486.8 2732.21  507.86 2747.47   516.3  2750.3   552.3 2768.61
#Mann= 5 ,-1 , 0
       0     .12       0   156.4     .04       0   195.6     .12       0
  455.38    .016       0  507.86     .12       0
Bank Sta=156.4,195.6
XS Rating Curve= 0 ,0
Exp/Cntr=0.3,0.1

Type RM Length L Ch R = 1 ,34485   ,542.2,551.2,558
XS GIS Cut Line= 3
     2125638.486      452172.821     2126067.753      452335.943
     2126290.973      452358.837
#Sta/Elev= 30
       0 2784.77      23 2774.27    45.9 2768.75    62.3 2762.52    85.3 2756.29
   121.4  2741.5   190.2  2720.3   203.4 2717.82   219.8 2711.47   249.3 2696.14
   275.5 2690.52   282.1 2687.71   295.2  2686.3   311.6 2685.56   341.1 2685.76
   347.7 2686.97   367.4 2691.55   390.3 2705.62   396.9 2707.26  415.53 2708.11
   429.7 2708.38   436.3 2711.47  447.12 2718.78   455.9 2722.66     469 2723.93
   517.8 2723.56   537.3 2724.97   576.3 2731.77   644.6 2746.05   683.6 2751.79
#Mann= 5 ,-1 , 0
       0     .12       0   295.2     .04       0   347.7     .12       0
  415.53    .016       0  447.12     .12       0
Bank Sta=295.2,347.7
XS Rating Curve= 0 ,0
Exp/Cntr=0.3,0.1

Type RM Length L Ch R = 1 ,33934   ,505.2,522.7,534.5
XS GIS Cut Line= 2
     2125443.884      452582.056     2125916.079      452951.226
#Sta/Elev= 30
       0 2755.05    22.9 2743.65    52.4 2727.24    68.8 2720.25    98.3 2713.16
   144.1 2708.57   173.6 2703.51   199.8  2693.5   212.9 2690.65   229.3 2688.95
   242.4  2683.5   258.8 2679.31   281.7 2678.57   317.7 2679.15   334.1 2679.13
   347.2 2688.16  351.05 2689.45  365.15 2691.36   386.5 2692.35   396.3 2687.99
  402.64 2686.64   419.2 2688.09   448.7 2698.98   474.9 2703.61   481.5 2705.83
   494.6 2712.66   527.3 2731.98   540.4 2742.17     547 2746.34   599.4  2770.5
#Mann= 6 ,-1 , 0
       0     .12       0   258.8     .04       0   317.7     .12       0
  351.05     .06       0  365.15    .016       0  402.64     .12       0
Bank Sta=258.8,317.7
XS Rating Curve= 0 ,0
Exp/Cntr=0.3,0.1

Type RM Length L Ch R = 1 ,33411   ,220.4,238.3,249.9
XS GIS Cut Line= 4
     2125179.515      452650.816     2125235.798      452964.754
     2125327.995      453193.395     2125518.823      453418.979
#Sta/Elev= 30
       0  2744.4    19.5 2736.88    35.8 2727.95    58.6 2724.78   104.1 2713.99
   143.2 2702.52   156.2 2700.93   169.2 2695.14     192 2689.58   257.1    2679
   406.5 2677.13   432.5  2675.7   448.7 2669.06   487.6 2668.49   503.8 2669.23
   513.6 2673.64     533 2690.02   539.5 2692.71   575.2 2696.27   597.9 2689.93
   604.4 2691.22   646.6 2721.49   662.9  2729.8   682.4 2751.43   695.4 2762.06
   711.6 2771.79   734.3 2781.23   773.3 2792.62   799.2 2802.71   860.9 2820.48
#Mann= 3 , 0 , 0
       0     .12       0   448.7     .04       0   503.8     .12       0
Bank Sta=448.7,503.8
XS Rating Curve= 0 ,0
Exp/Cntr=0.3,0.1

Type RM Length L Ch R = 1 ,33173   ,514.8,507,483.2
XS GIS Cut Line= 4
     2125089.023      452622.121     2125091.885      452971.259
      2125051.82      453214.511     2125097.608      453506.413
#Sta/Elev= 30
       0 2775.69    22.8 2764.65      49 2744.62    71.8 2734.11   117.5  2724.6
   172.9 2708.82   231.7 2698.52   264.3 2688.16   349.2 2672.37   358.9 2667.98
   391.3 2670.49   417.3 2667.86     440 2669.81  473.19 2668.73   488.6 2667.93
   514.6 2666.36     534 2666.73   540.5 2669.02   556.8 2690.25   563.2  2696.1
  652.72 2713.08   670.4 2706.82   699.6 2707.55  712.52 2716.22   735.3 2739.09
     758 2748.25   780.8 2779.85   793.7 2791.16   832.7 2808.35   891.2 2827.06
#Mann= 6 ,-1 , 0
       0     .12       0  473.19     .08       0   488.6     .04       0
   540.5     .12       0  652.72    .016       0  712.52     .12       0
#XS Ineff= 2 , 0
           392.8 2691.33
Permanent Ineff=
       F       F
Bank Sta=488.6,540.5
XS Rating Curve= 0 ,0
Exp/Cntr=0.3,0.1

Type RM Length L Ch R = 1 ,32666   ,318.7,316.1,309.6
XS GIS Cut Line= 2
2124467.14291861452803.0957368082124783.74554999453622.041209973
#Sta/Elev= 30
       0 2794.17    89.2 2751.98   117.3  2739.9   145.4 2730.11   215.8 2710.08
   342.4 2687.41     360 2679.44   381.1 2666.42   395.2 2660.59   422.22656.665
   429.6 2655.09   444.4    2655   472.7 2655.06   480.3 2656.29   497.2  2664.2
   511.3 2665.64   528.9 2665.36   553.5 2671.56     564 2676.84   581.6 2682.15
   613.3 2689.22   648.5  2694.7   666.1  2703.5   680.1 2705.02   709.7 2705.34
   743.4 2726.98   773.3 2742.15   813.8 2759.58   855.8 2773.71     878 2785.44
#Mann= 3 , 0 , 0
       0     .12       0   422.2     .04       0   480.3     .12       0
Bank Sta=422.2,480.3
XS Rating Curve= 0 ,0
Exp/Cntr(USF)=0,0
Exp/Cntr=0.3,0.1

Type RM Length L Ch R = 1 ,32350   ,545,552.3,558.9
XS GIS Cut Line= 2
     2124181.837      453042.804     2124545.284       453726.77
#Sta/Elev= 30
       0 2742.87    26.1 2728.17    62.1 2711.65    71.9 2709.38      85 2702.86
   130.7 2687.87   143.8 2686.62   163.4 2680.55   189.6    2675   251.6 2667.13
   271.2 2661.44   290.9  2659.2     317 2650.84   330.1 2649.48   375.8 2650.67
   395.4 2660.03   411.8 2661.99   428.1  2668.6   447.7 2670.66   516.4 2684.25
     536 2690.75  559.29 2691.45  592.74 2692.23   601.3    2694   620.9  2708.5
   647.1 2716.43   663.4 2723.74   692.8 2733.76   751.7 2758.35   774.5 2769.29
#Mann= 5 ,-1 , 0
       0     .12       0     317     .04       0   375.8     .12       0
  559.29    .016       0  592.74     .12       0
Bank Sta=317,375.8
XS Rating Curve= 0 ,0
Exp/Cntr=0.3,0.1

Type RM Length L Ch R = 1 ,31797   ,491.9,489.2,480.9
XS GIS Cut Line= 2
2123749.51028749453166.1334207882123943.69323473454014.628472882
#Sta/Elev= 30
       0  2780.1    17.6 2769.63    28.6 2766.05    39.5 2757.07    61.4 2744.58
   207.7 2680.43   221.1 2678.25   228.5 2673.82   248.1 2665.53   268.2 2660.99
   307.9  2655.2   328.8 2648.49   342.3 2646.46   359.1 2640.59   382.7 2640.06
     413  2640.7   418.9  2642.7   429.8 2649.55   436.5 2651.21   483.2  2652.9
   510.6 2652.28   527.4 2655.21   557.7 2657.44   604.8 2658.89   621.6  2663.6
     662 2663.98   678.9 2665.69   793.3 2686.39   823.6 2695.05   870.4 2711.54
#Mann= 3 , 0 , 0
       0     .12       0   359.1     .04       0     413     .12       0
Bank Sta=359.1,413
XS Rating Curve= 0 ,0
Exp/Cntr(USF)=0,0
Exp/Cntr=0.3,0.1

Type RM Length L Ch R = 1 ,31308   ,625.9,670.9,694.7
XS GIS Cut Line= 2
     2123271.789      453400.527     2123620.927      454198.965
#Sta/Elev= 30
       0 2702.86   108.1 2675.97   137.6  2674.5   180.2 2668.36   193.3 2668.48
   209.7 2665.63   258.8 2662.13   288.3 2654.21   298.1 2646.65   311.2 2639.52
   330.9 2634.25   373.5 2633.51  384.81 2634.28     403 2641.77   419.3 2643.85
     439 2643.47   452.1 2640.88   494.7 2647.32   524.2 2646.35   567.7 2649.44
  599.94 2652.29   609.4 2650.83   625.7 2655.97   651.9 2658.83  684.11 2659.63
  696.65 2660.62  757.83 2663.49  793.36 2664.88  831.56 2670.84   871.4 2681.54
#Mann= 10 ,-1 , 0
       0     .12       0   330.9     .04       0  384.81     .12       0
   567.7    .016       0  599.94     .12       0  684.11    .016       0
  696.65     .12       0  757.83    .016       0  793.36     .12       0
  831.56    .016       0
Bank Sta=330.9,384.81
XS Rating Curve= 0 ,0
Exp/Cntr=0.3,0.1

Type RM Length L Ch R = 1 ,30637   ,822.9,808.3,788.9
XS GIS Cut Line= 3
     2123045.708      453122.934     2122894.033      453618.022
     2122573.513      453958.575
#Sta/Elev= 30
       0  2801.5    42.6 2783.01    68.8 2769.16   124.5 2751.19   160.6 2736.48
   173.7 2729.45   190.1 2724.08   239.2 2701.72   357.2 2652.86   370.3 2650.49
   403.1 2640.44   432.6 2635.74     544 2635.12     593 2626.93   619.2 2626.04
   661.7 2625.13   681.3 2626.67   691.1 2631.96   704.2 2634.83     714 2639.05
   730.3 2640.35   756.5 2641.64  771.18 2650.81   792.5  2667.4   884.1 2676.64
   916.8 2682.77   939.7 2683.48   952.8 2688.19   962.6 2689.57   985.5 2701.74
#Mann= 5 ,-1 , 0
       0     .12       0   619.2     .04       0   681.3     .12       0
   730.3    .016       0  771.18     .12       0
Bank Sta=619.2,681.3
XS Rating Curve= 0 ,0
Exp/Cntr=0.3,0.1

Type RM Length L Ch R = 1 ,29829   ,650.7,639.3,623.8
XS GIS Cut Line= 2
     2122267.302      452713.698     2122081.286      453735.356
#Sta/Elev= 30
       0 2840.33    42.6 2821.77    65.5 2809.88   121.2  2787.3   144.1 2776.22
   196.6 2760.56   245.7 2740.01   324.3 2718.48   396.4 2694.51   442.2  2685.8
   481.6 2675.07   494.7 2668.35   507.8 2657.67   524.1 2652.38   563.4 2616.81
   576.6 2611.28   612.6 2610.11   645.4 2611.21     665 2616.31   687.9    2617
     701 2620.49   733.8 2620.71  746.48 2626.11   776.5 2625.67     796 2623.83
   822.2 2636.49   884.5 2652.52   966.4 2668.31   979.5 2669.25  1038.4    2684
#Mann= 5 ,-1 , 0
       0     .12       0   576.6     .04       0   645.4     .12       0
  746.48    .016       0   776.5     .12       0
Bank Sta=576.6,645.4
XS Rating Curve= 0 ,0
Exp/Cntr=0.3,0.1

Type RM Length L Ch R = 1 ,29190   ,768.4,778.3,788.9
XS GIS Cut Line= 4
     2121497.482      452659.324     2121503.206      453248.852
      2121557.58      453500.689     2121603.368      453784.006
#Sta/Elev= 30
       0 2793.98    22.9  2783.9    32.8 2781.15    72.1 2771.89    91.7 2770.35
     167 2752.11   252.2 2723.73   396.3 2683.56   425.8 2677.18   507.7 2649.46
   563.4 2634.32   599.3 2631.15   648.3 2622.17   677.6 2601.16   723.3 2600.03
   746.1 2601.09   762.4 2607.05     795 2607.51   811.3 2613.94  823.62 2614.41
   843.9 2613.97  853.77 2616.86     870 2626.31   879.8 2634.55   886.3 2636.42
     945 2645.11   967.9 2647.08   980.9 2654.08  1088.5  2677.1  1134.2 2690.82
#Mann= 5 ,-1 , 0
       0     .12       0   677.6     .04       0   746.1     .12       0
  823.62    .016       0  853.77     .12       0
Bank Sta=677.6,746.1
XS Rating Curve= 0 ,0
Exp/Cntr=0.3,0.1

Type RM Length L Ch R = 1 ,28411   ,841.5,829,800.6
XS GIS Cut Line= 3
     2120867.889      452659.324      2120804.93      453211.649
     2120739.109      453712.461
#Sta/Elev= 30
       0 2891.05    68.7 2855.96    94.8 2816.55   134.1 2798.34   179.8 2771.37
   232.2 2749.88     278 2726.12   294.3 2714.28   353.2 2687.88   372.8 2682.02
   454.5 2646.75   523.2 2625.31   539.6 2617.16   555.9 2604.82   578.9 2594.28
   598.5 2590.26   618.2 2593.03   726.5  2592.6   739.6 2586.81     756 2585.49
   805.2 2586.55     815 2593.79   834.7 2596.67   847.8 2604.95   906.9 2612.73
   926.5 2612.55  943.36 2619.35   992.1 2619.69 1002.94  2623.4    1061  2633.8
#Mann= 5 ,-1 , 0
       0     .12       0   739.6     .04       0   805.2     .12       0
  943.36    .016       0 1002.94     .12       0
#XS Ineff= 2 , 0
          619.57 2596.15
Permanent Ineff=
       F       F
Bank Sta=739.6,805.2
XS Rating Curve= 0 ,0
Exp/Cntr=0.3,0.1

Type RM Length L Ch R = 1 ,27582   ,863.1,876.4,885.9
XS GIS Cut Line= 4
     2119869.126      453028.495     2119983.598      453497.827
     2120138.134       453758.25     2120172.475      453915.648
#Sta/Elev= 30
       0 2777.25    39.2 2761.58    81.6 2747.72   166.5 2699.99   215.4 2678.89
   267.7 2660.28   352.5 2635.29   372.1 2626.54   424.3 2606.92   486.4 2594.81
   515.6  2582.5   525.4 2579.89   613.3 2575.55   623.1    2574   636.1 2569.54
   645.9 2568.58   681.7 2569.48     711 2571.83   727.3  2574.7   750.1 2573.13
   759.9 2577.15  768.74 2583.53   782.7  2591.3   818.1 2590.72  831.26 2595.07
   850.4 2606.09   872.9 2622.17   882.6 2626.88   905.1 2632.96     947 2638.79
#Mann= 5 ,-1 , 0
       0     .12       0   636.1     .04       0   681.7     .12       0
  768.74    .016       0  831.26     .12       0
Bank Sta=636.1,681.7
XS Rating Curve= 0 ,0
Exp/Cntr=0.3,0.1

Type RM Length L Ch R = 1 ,26706   ,494.7,495.5,487.1
XS GIS Cut Line= 4
     2119176.574      453297.502      2119233.81      453663.811
      2119250.98      453941.404     2119302.493      454176.071
#Sta/Elev= 30
       0 2755.33    45.5 2728.47   104.1 2699.34   120.3  2692.6   143.1 2678.74
   175.6 2662.65   208.1 2647.49   256.9 2629.98   279.7 2613.87   305.7 2600.32
   354.5 2587.45   403.5 2579.06   429.6  2571.9   449.3 2569.41   475.5  2559.6
   491.8 2558.15   547.4 2558.33   557.3 2559.52   576.9 2564.84   632.5 2566.32
   639.1 2568.92  657.93 2580.85  705.43 2582.85   726.8 2595.91   739.8 2598.24
     756 2604.13   778.7 2608.64   788.5  2612.4   853.4 2617.16   889.1 2624.75
#Mann= 5 ,-1 , 0
       0     .12       0   475.5     .04       0   557.3     .12       0
  657.93    .016       0  705.43     .12       0
Bank Sta=475.5,557.3
XS Rating Curve= 0 ,0
Exp/Cntr=0.3,0.1

Type RM Length L Ch R = 1 ,26211   ,624.5,627.4,622.3
XS GIS Cut Line= 2
2118650.09723808453259.0035259932118848.50155375454318.566999006
#Sta/Elev= 30
       0 2837.63    31.4 2819.88    54.7 2800.92    74.7 2777.64   121.5 2742.58
   134.8 2735.99   151.5 2721.82   191.6 2701.65   271.1 2647.05   328.4  2622.7
   375.2 2612.93   428.5 2589.59   498.8 2571.64   525.4 2568.64   548.7 2561.54
   558.7 2554.65   565.4 2552.34   618.8 2551.71   638.8 2553.71   655.5 2560.89
   695.8  2559.7   715.3  2564.9     749 2567.78   805.7 2572.38   855.8  2572.9
   869.2 2578.04   969.3 2592.41   982.6 2597.25  1029.4 2605.26    1078 2617.86
#Mann= 3 , 0 , 0
       0     .12       0   558.7     .04       0   638.8     .12       0
Bank Sta=558.7,638.8
XS Rating Curve= 0 ,0
Exp/Cntr(USF)=0,0
Exp/Cntr=0.3,0.1

Type RM Length L Ch R = 1 ,25583   ,682,668.9,646
XS GIS Cut Line= 2
     2118051.892       453549.34     2118277.973      454465.111
#Sta/Elev= 30
       0 2723.23    45.8  2707.8    91.7 2689.53   137.6 2675.46   183.4 2655.95
   242.4 2626.06   307.9 2597.04   327.5 2581.05   343.9 2564.78   353.7 2557.66
   376.6 2550.72   386.5 2546.05   422.5 2544.84   458.5 2545.92   471.6 2552.57
   484.7 2554.62   510.9 2553.47     524 2555.68     547 2555.87   622.3 2553.39
   638.7 2554.33  656.34 2552.58   671.4 2556.59  686.76 2557.31   707.4 2557.15
  717.18 2553.72   740.2 2553.34   805.7 2567.91   864.7  2585.8   943.3 2613.11
#Mann= 6 ,-1 , 0
       0     .12       0   386.5     .04       0   458.5     .12       0
  656.34     .08       0  686.76    .016       0  717.18     .12       0
Bank Sta=386.5,458.5
XS Rating Curve= 0 ,0
Exp/Cntr=0.3,0.1

Type RM Length L Ch R = 1 ,24914   ,249.7,229.8,201.1
XS GIS Cut Line= 4
     2117253.454      453763.973     2117445.194      454058.737
     2117576.836      454196.103     2117948.868      454445.078
#Sta/Elev= 30
       0 2804.12   104.2 2734.97   136.8 2710.87   159.5 2691.58   182.3 2680.13
   205.1 2664.53   227.9 2652.56   273.5 2634.31   299.5 2621.28   381.2  2591.7
   404.1 2574.56   427.1 2547.23   436.9 2540.69   466.4 2539.01   505.8 2540.51
   522.2 2546.76   532.1 2548.06   666.1 2549.13   721.6    2546  737.15 2548.22
   754.3 2552.33  790.25 2553.65     800  2553.5   829.4 2545.87   875.2 2550.46
   937.3 2547.66   956.9    2554   966.7 2560.62     983 2562.21   989.6 2565.35
#Mann= 5 ,-1 , 0
       0     .12       0   436.9     .04       0   505.8     .12       0
  737.15    .016       0  790.25     .12       0
#XS Ineff= 2 , 0
                          613.04         2549.14
Permanent Ineff=
       F       F
Bank Sta=436.9,505.8
XS Rating Curve= 0 ,0
Exp/Cntr=0.5,0.3

Type RM Length L Ch R = 1 ,24684   ,307.5,321.3,338.6
XS GIS Cut Line= 4
     2116915.763       453869.86     2117167.601      454224.721
     2117450.917      454299.127     2117931.697      454482.282
#Sta/Elev= 30
       0 2676.03    52.4 2672.84      72 2668.11     121 2665.44   176.7 2653.66
   235.6 2634.77   320.6 2618.51   366.4 2597.95   422.1 2576.34   467.7 2567.76
   490.5  2560.4     523 2555.79   542.6 2546.18   568.6 2539.66   578.4 2538.44
   659.7 2540.06   679.2 2546.63     787 2544.91  826.67 2548.93   865.7 2551.01
  909.64 2552.53   934.5 2552.17     964 2544.22  1000.1 2546.96    1082 2544.66
  1127.9 2551.52  1173.7 2566.91    1200 2567.37  1219.6 2579.54  1242.6 2585.88
#Mann= 6 ,-1 , 0
       0     .12       0   568.6     .04       0   659.7     .12       0
  826.67     .08       0   865.7    .016       0  909.64     .12       0
#XS Ineff= 2 , 0
                             680         2548.83
Permanent Ineff=
       F       F
Bank Sta=568.6,659.7
XS Rating Curve= 0 ,0
Exp/Cntr=0.5,0.3

Type RM Length L Ch R = 1 ,24363   ,394.6,409.6,438.4
XS GIS Cut Line= 4
      2116397.78      454041.567     2116978.723      454410.737
     2117187.633      454525.208     2117542.495      454751.289
#Sta/Elev= 30
       0 2637.32    26.2 2631.13   121.3 2593.83   170.4 2583.86   216.3 2580.58
   262.2 2569.66   301.6 2567.86   327.8 2554.35   344.2 2549.17   380.2  2554.4
   426.1 2541.98   462.2 2540.82  490.61 2544.63   563.8  2542.1  600.75  2546.5
  655.82 2547.06   678.5 2541.79   701.4 2540.21   773.2 2541.65   786.2 2537.07
     845 2537.28   867.8 2535.99   887.4 2536.46   903.7 2543.67  1187.5 2541.61
  1210.3  2552.7  1285.3 2577.61  1314.7 2594.24    1331 2596.54  1347.3  2607.9
#Mann= 6 ,-1 , 0
       0     .12       0  490.61     .08       0  600.75    .016       0
  655.82     .12       0   786.2     .04       0     845     .12       0
#XS Ineff= 2 , 0
          767.04 2543.92  902.67         2544.31
Permanent Ineff=
       F       F
Bank Sta=786.2,845
XS Rating Curve= 0 ,0
Exp/Cntr=0.5,0.3

Type RM Length L Ch R = 1 ,23954   ,464.5,457.2,457.8
XS GIS Cut Line= 4
     2116449.292      454098.802     2116778.398      454636.818
      2116798.43      454828.558     2116786.983      454991.679
#Sta/Elev= 30
       0 2602.95      36  2588.5    78.4 2577.65   114.4  2568.8   176.5 2557.98
   215.7 2534.98  241.37 2534.91   261.4 2542.32  310.62 2541.09   336.6 2539.96
  345.24 2536.45   352.9 2533.31   372.5 2532.47   392.1 2536.68   424.8 2533.14
   473.8  2537.3     549 2537.69   578.4 2532.33   594.7 2534.56     647  2536.3
   705.8 2530.49     732 2529.63  750.53 2530.75     781 2541.07   794.1 2552.63
   807.1 2569.22   820.2 2581.32   856.2 2598.81   954.3 2652.84     987  2682.7
#Mann= 6 ,-1 , 0
       0     .12       0  241.37     .08       0  310.62    .016       0
  345.24     .12       0   705.8     .04       0  750.53     .12       0
#XS Ineff= 2 , 0
          267.39 2543.73
Permanent Ineff=
       F       F
Bank Sta=705.8,750.53
XS Rating Curve= 0 ,0
Exp/Cntr=0.3,0.1

Type RM Length L Ch R = 1 ,23496   ,502,475.6,458.5
XS GIS Cut Line= 4
     2116386.333      454084.493     2116366.301      454496.591
     2116369.162      454674.021     2116386.333      454925.858
#Sta/Elev= 30
       0 2620.54      36 2604.95    62.2 2599.73   108.1  2585.1   163.7 2570.08
   170.3 2566.62   186.6 2552.28   222.7 2531.22     239 2529.88  279.61 2531.15
     298 2537.91  309.18 2538.15  338.76 2534.91   363.5 2529.91   386.4 2527.78
   425.5 2527.14   444.8 2528.84   457.8 2525.07   464.2 2524.14   515.8 2524.42
   525.5  2525.6   541.6 2532.05   586.8 2531.51   606.4 2535.49     649 2534.22
   665.4 2537.21   724.4 2561.28     754 2569.14   809.7 2590.76   842.5 2609.55
#Mann= 6 ,-1 , 0
       0     .12       0  279.61     .08       0  309.18    .016       0
  338.76     .12       0   457.8     .04       0   525.5     .12       0
#XS Ineff= 2 , 0
          318.26 2537.64
Permanent Ineff=
       F       F
Bank Sta=457.8,525.5
XS Rating Curve= 0 ,0
Exp/Cntr=0.3,0.1

Type RM Length L Ch R = 1 ,23021   ,524.2,510.6,507.2
XS GIS Cut Line= 3
     2115736.708      454508.038      2116028.61      454811.387
     2116263.276      455046.053
#Sta/Elev= 30
       0 2663.03      13 2653.88    22.8 2650.06    65.3 2626.08   104.4 2601.08
     111 2595.32   127.3 2576.71   137.1 2567.48   150.1 2561.04   169.7 2547.47
   189.3 2529.69   199.1 2527.38   225.2 2527.75  250.69 2531.05  291.68 2528.03
   306.8  2519.3   345.9 2518.24   368.8 2519.67   378.6 2525.42   381.8 2525.79
   505.6  2524.3   518.6 2525.22   544.6 2523.73   570.6 2525.64   586.9 2529.94
   632.5 2529.91   648.7 2535.46   661.8 2543.94   681.3 2552.54   752.8 2594.76
#Mann= 5 ,-1 , 0
       0     .12       0  250.69    .016       0  291.68     .12       0
   306.8     .04       0   368.8     .12       0
#XS Ineff= 2 , 0
                          520.07         2524.87
Permanent Ineff=
       F       F
Bank Sta=306.8,368.8
XS Rating Curve= 0 ,0
Exp/Cntr=0.3,0.1

Type RM Length L Ch R = 1 ,22510   ,572.6,615.3,656.2
XS GIS Cut Line= 4
     2115433.359      454943.029     2115690.919      455177.696
      2115868.35      455269.273     2116174.561      455352.264
#Sta/Elev= 30
       0  2647.3    22.8  2638.4    58.6 2620.12   110.7 2605.96   136.8 2594.37
   146.5 2586.86   162.8 2569.87   182.4 2554.76   201.9 2543.18   214.9 2528.18
  226.25 2524.05  266.21 2524.89   283.3 2523.02   302.8 2516.49     391 2518.66
   400.8 2514.59   453.2 2513.56   489.2 2514.68   502.3 2519.56   564.5 2516.76
   603.7 2523.91   636.4 2524.55   649.5 2532.02   665.8 2547.02   695.3 2562.29
   724.7 2574.61   760.7 2581.77   783.6 2590.52   835.9 2623.78   865.4 2639.53
#Mann= 5 ,-1 , 0
       0     .12       0  226.25    .016       0  266.21     .12       0
   400.8     .04       0   489.2     .12       0
#XS Ineff= 2 , 0
          383.57  2518.7  526.08         2518.82
Permanent Ineff=
       F       F
Bank Sta=400.8,489.2
XS Rating Curve= 0 ,0
Exp/Cntr=0.3,0.1
